--- 6888_ras.prj (project) ---

Proj Title=6888
Current Plan=p01
Default Exp/Contr=0.3,0.1
English Units
Geom File=g01
Flow File=f01
Plan File=p01
Y Axis Title=Elevation
X Axis Title(PF)=Main Channel Distance
X Axis Title(XS)=Station
BEGIN DESCRIPTION:
RFD model 6888 exported to HEC-RAS
END DESCRIPTION:

--- 6888_ras.p01 (plan) ---

Plan Title=Plan 01
Program Version=4.10
Short Identifier=Plan 01
Geom File=g01
Flow File=f01
Subcritical Flow
Calc Critical at every XS
Secant Critical Depth

--- 6888_ras.f01 (steady flow) ---

Flow Title=Flow 01
Program Version=5.01
Number of Profiles= 6
Profile Names=10yr,25yr,50yr,100yr,100plus,500yr
River Rch & RM=6888,39,15705.05
  751.85 1307.87  1867.1 2425.13  3540.7  5407.1
River Rch & RM=6888,39,15465.04
  754.61 1312.86  1874.4 2434.82 3554.83 5426.62
River Rch & RM=6888,39,15225.03
     757 1317.17 1880.72  2443.2 3567.07 5443.52
River Rch & RM=6888,39,14985.02
  761.78 1325.81 1893.36 2459.96 3591.55 5477.25
River Rch & RM=6888,39,   14745
  767.45 1336.07 1908.38  2479.9 3620.65 5517.36
River Rch & RM=6888,39,14504.99
  769.65 1340.04 1914.19 2487.61 3631.91 5532.86
River Rch & RM=6888,39,14264.98
  777.69 1354.57 1935.47 2515.84 3673.12 5589.53
River Rch & RM=6888,39,14024.97
  782.93 1364.08 1949.41 2534.35 3700.15 5626.76
River Rch & RM=6888,39,13544.95
  793.93  1384.1 1978.86 2573.58 3757.42 5706.03
River Rch & RM=6888,39,13304.94
  795.33 1386.67 1982.64 2578.61 3764.78 5716.23
River Rch & RM=6888,39,13064.93
  796.21 1388.27    1985 2581.76 3769.37  5722.6
River Rch & RM=6888,39,12824.92
  798.67 1392.75  1991.6 2590.57 3782.23 5740.42
River Rch & RM=6888,39,12584.91
  805.34 1404.92 2009.52 2614.46 3817.11 5788.68
River Rch & RM=6888,39,12288.86
 1006.49 1769.76 2544.96 3326.23 4856.29 7189.55
River Rch & RM=6888,39,12064.45
 1006.83 1770.37 2545.86 3327.42 4858.04 7191.87
River Rch & RM=6888,39,11840.05
 1012.57 1780.88 2561.39 3348.18 4888.35 7232.58
River Rch & RM=6888,39,11762.94
 1013.06 1781.78 2562.72 3349.96 4890.94 7236.07
River Rch & RM=6888,39,11434.08
 1142.19 2019.82  2915.7 3823.42 5582.19 8162.32
River Rch & RM=6888,39,10989.97
 1175.15 2080.06 3004.58  3942.1 5755.47 8389.31
River Rch & RM=6888,39,10563.34
 1178.06 2085.36 3012.37 3952.49 5770.63 8409.02
River Rch & RM=6888,39,10242.18
 1188.51  2104.4 3040.43 3989.89 5825.25 8480.08
River Rch & RM=6888,39,10064.62
 1189.64 2106.46 3043.46 3993.93 5831.14 8487.72
River Rch & RM=6888,39,9179.738
 1258.23 2230.77 3225.91 4236.42 6185.18 8942.29
River Rch & RM=6888,39,8584.131
 1307.94 2321.24 3359.08 4413.84  6444.2 9274.43
River Rch & RM=6888,39,8090.633
 1310.52 2325.91 3365.92 4422.93 6457.48 9291.29
River Rch & RM=6888,39,7597.136
 1329.48 2360.33  3416.5 4490.22 6555.71 9416.25
River Rch & RM=6888,39,7103.638
 1335.09 2370.49 3431.41 4510.03 6584.64 9452.88
River Rch & RM=6888,39,6610.141
 1485.14 2640.22 3825.35 5031.17 7345.5110397.86
River Rch & RM=6888,39,6116.643
  1511.8 2688.63 3896.53 5125.88 7483.7810570.57
River Rch & RM=6888,39,5623.146
 3497.95 6140.22 8829.79 11517.616815.69 20766.7
River Rch & RM=6888,39,5129.648
 3503.56 6150.47 8844.9311537.7916845.17 20799.7
River Rch & RM=6888,39,4636.151
 3509.12 6160.66    886011557.9116874.5420832.68
River Rch & RM=6888,39,4142.654
 3536.44  6210.9 8934.4211657.4817019.9220996.52
River Rch & RM=6888,39,1554.245
 3831.89 6746.72 9721.8512703.2318546.7222675.19
River Rch & RM=6888,39,1434.017
  3834.1  6750.8 9727.9312711.3918558.6322688.54
River Rch & RM=6888,39,1287.098
 3835.07  6752.6 9730.61   1271518563.8922694.47
River Rch & RM=6888,39, 60.2721
 3888.87 6852.37 9879.2212914.73 18855.523021.98
Boundary for River Rch & Prof#=6888,39,1
Up Type= 0
Dn Type= 2
Boundary for River Rch & Prof#=6888,39,2
Up Type= 0
Dn Type= 2
Boundary for River Rch & Prof#=6888,39,2
Up Type= 0
Dn Type= 2
Boundary for River Rch & Prof#=6888,39,2
Up Type= 0
Dn Type= 2
Boundary for River Rch & Prof#=6888,39,2
Up Type= 0
Dn Type= 2
Boundary for River Rch & Prof#=6888,39,2
Up Type= 0
Dn Type= 2

--- 6888_ras.g01 (geometry) ---

Geom Title=6888
Program Version=4.10

River Reach=6888,39
Reach XY= 30
803996.569285393720598.832955236803510.127665462720189.462546531
802374.308772684720117.872198572801098.267105996719476.379143027
800885.593494893 719274.99025414800901.218494895 719017.17775413
800812.120926711718589.479903866801110.992672592718472.116187903
801090.454878748718321.295123822801182.008487525718191.464654441
801211.424298525 717907.68955863801428.006001304717736.741176821
801687.675173401717326.125812788802160.186480851717063.166614601
802329.169883788716885.233309702802786.523796445 715926.58492682
803056.221917213715550.914546142803297.919883759715393.045809687
 803482.73369694715155.589534496804021.424732955714088.068894999
804228.475439313 713090.09442082804640.801828239712714.226365238
804562.676828238712445.997198571804751.044883788712427.768031904
804926.999874176712192.983625298805092.448787692711776.702904273
805093.926828237710834.886087459805221.010161549710019.955531906
805103.822661582709371.518031922804991.261902662709108.636674657

Type RM Length L Ch R = 1 ,15705.05,240.010900,240.010900,240.010900
XS GIS Cut Line= 6
804275.183353226720249.041324006804080.470332884720485.947639584
804021.321643071 720560.62352682803970.434827411 720636.22268059
803862.458689903720781.166639784803837.842385789720815.778224701
#Sta/Elev= 30
9552.517160.68449584.304149.10339599.063141.93829624.951132.6063 9650.84 127.578
9676.728125.38839689.672122.77369726.046122.62199780.282120.92529883.478125.8293
9916.301126.52679947.262125.63899965.668124.57769996.026112.862610001.35111.6978
10008.02111.883410020.05119.548510032.07 123.212 10044.1124.104110068.98124.1052
10081.45115.636610088.14 115.82510104.88122.772910131.33 129.611 10143.8129.5205
10156.27 136.31410171.84139.846410188.58 145.91410255.56176.436310268.78 179.427
#Mann= 3 , 0 , 0
9552.517    0.04       09552.517    0.04       010268.78    0.04       0
#XS Ineff= 2 , 0
       0                               0
Bank Sta=9552.517,10268.78
Exp/Cntr=0.3,0.1

Type RM Length L Ch R = 1 ,15465.04,240.011000,240.011000,240.011000
XS GIS Cut Line= 6
804148.478022107720011.205371697804058.560249719720127.633342966
803862.287644138720375.909759978803816.417358279720440.182458158
803781.559615921720490.645451122803690.334103136720616.014442827
#Sta/Elev= 30
9456.443149.87819499.143128.94469511.214125.67889527.574123.91549549.683119.7334
9587.588117.40799612.941117.34039625.688116.16489651.183115.34519722.165118.7559
9740.415118.26039753.162118.84659829.646116.34859851.164117.36879867.289115.1677
9899.539116.19939943.491116.27329955.776 114.9869968.062115.21279992.633106.6571
10004.84107.7536 10036.7115.999810054.28116.080510065.72122.673410088.48138.9835
10102.82141.320910127.55155.314710164.66164.107910201.76167.480710215.38167.9672
#Mann= 3 , 0 , 0
9456.443    0.04       09456.443    0.04       010215.38    0.04       0
#XS Ineff= 2 , 0
       0                               0
Bank Sta=9456.443,10215.38
Exp/Cntr=0.3,0.1

Type RM Length L Ch R = 1 ,15225.03,240.010900,240.010900,240.010900
XS GIS Cut Line= 6
803852.047859409720012.652208113803721.712230671720190.798262858
803683.941637779720234.868907631803573.657192161720350.063685889
803520.416822842720422.931327268803496.747914985720463.877216307
#Sta/Elev= 30
9641.633145.86289654.252144.16979671.553137.97029693.405138.55379705.895137.5625
9730.309128.96219757.408117.67269767.213114.59359774.579113.70939791.816112.7798
9816.897  113.589842.331112.6206 9903.47113.2314 9934.57111.60259948.494109.4619
9962.055108.62719976.342106.0661    9999105.227110005.06105.554510019.24107.8941
 10046.2109.106610063.04111.661610086.23117.332810124.29120.432110136.55120.7717
10148.62123.487810162.08131.425510172.65135.3937 10184.2 138.21810217.56140.7293
#Mann= 3 , 0 , 0
9641.633    0.04       09641.633    0.04       010217.56    0.04       0
#XS Ineff= 2 , 0
       0                               0
Bank Sta=9641.633,10217.56
Exp/Cntr=0.3,0.1

Type RM Length L Ch R = 1 ,14985.02,240.011000,240.011000,240.011000
XS GIS Cut Line= 6
803456.063954501720034.131485344803435.190389022720134.165610475
803412.788902365720279.756481913803399.502756474720342.534683216
803385.770638951720396.858495363803343.858309315720535.448967888
#Sta/Elev= 30
9856.583137.84119888.346130.4377 9898.55126.06889918.916114.22669929.099111.1646
9949.464108.80569959.642108.49419969.757107.00329979.872 107.3889989.987103.9614
 10000.1 102.90110010.22103.374410030.46102.471410050.69102.738510060.81105.3834
10081.05104.465110101.29106.441910111.46108.737910142.13112.627310152.35116.2387
10162.57118.801310172.81120.430810193.44120.277810203.76122.479510224.39123.6052
10245.21132.352310276.46133.405210307.72136.903210339.08141.332810371.11144.6465
#Mann= 3 , 0 , 0
9856.583    0.04       09856.583    0.04       010371.11    0.04       0
#XS Ineff= 2 , 0
       0                               0
Bank Sta=9856.583,10371.11
Exp/Cntr=0.3,0.1

Type RM Length L Ch R = 1 ,   14745,240.010900,240.010900,240.010900
XS GIS Cut Line= 6
 803217.60739516720013.037791822803209.265996373720149.445748313
803205.424740154720172.908835479803194.670006033720215.142375789
803188.466445567720247.694997234803164.049178799720440.441172926
#Sta/Elev= 30
9817.769129.53899819.735129.37549829.753126.69039839.772121.69299859.809114.0153
9879.847107.86289889.865106.25729909.903104.92169939.959104.02959949.977101.2657
 9960.0699.1574210001.0196.6413210021.65101.886810031.83105.298110042.01112.4771
10052.19115.811110062.29 114.71910082.44117.861810092.52118.135110102.59120.3949
10112.67120.515710122.74119.889210132.81 122.32610142.89 123.85610163.04128.0729
10173.11129.727610193.26134.731310203.34137.811810223.49142.242810249.23145.4988
#Mann= 3 , 0 , 0
9817.769    0.04       09817.769    0.04       010249.23    0.04       0
#XS Ineff= 2 , 0
       0                               0
Bank Sta=9817.769,10249.23
Exp/Cntr=0.3,0.1

Type RM Length L Ch R = 1 ,14504.99,240.011000,240.011000,240.011000
XS GIS Cut Line= 6
802978.895291188 719959.80815053 802970.58179045720107.286946587
 802964.48935562720157.945654171802959.250751952720202.203104752
802954.327663995720325.576753621802952.223905341720358.388566042
#Sta/Elev= 30
9802.262119.46489807.462119.54869817.478117.1978 9837.51114.66419847.526113.7262
9857.542113.83449887.589110.11569897.605110.26879917.637108.39529927.653 106.829
9937.669104.15189967.81399.659899977.88496.779799987.95494.529759998.02594.93931
 10008.194.2704610018.1795.5022310028.24 95.447310038.3196.2787410048.3799.71667
10058.37 104.23310078.39111.8238 10088.4112.981110118.42117.917610128.43121.2488
10138.44121.753910148.45123.956210178.48128.0928 10188.5127.546510201.92128.4172
#Mann= 3 , 0 , 0
9802.262    0.04       09802.262    0.04       010201.92    0.04       0
#XS Ineff= 2 , 0
       0                               0
Bank Sta=9802.262,10201.92
Exp/Cntr=0.3,0.1

Type RM Length L Ch R = 1 ,14264.98,240.010900,240.010900,240.010900
XS GIS Cut Line= 6
802764.681850261719910.821805768802743.085021119720114.874874913
802737.510092756720146.030166994802724.534504125720199.310208366
 802716.88580985720238.002641099802702.883496582720330.502587533
#Sta/Elev= 30
9734.481106.33099758.794103.1702 9768.85102.15749788.961101.24599809.07399.43794
9839.24198.647289859.35297.404089869.40897.09239 9889.5297.634299899.57697.75328
9909.63296.346079919.68893.683029939.80194.593189949.95994.439399960.11895.24621
9970.27793.044529980.54892.292159990.83290.6372310001.1389.2263910011.4390.39155
10021.7293.3311610042.16101.981910052.35104.568410072.68106.258910103.02107.9337
10113.14109.573710133.36111.848910143.48 113.40310153.59115.300810159.16114.7213
#Mann= 3 , 0 , 0
9734.481    0.04       09734.481    0.04       010159.16    0.04       0
#XS Ineff= 2 , 0
       09880.029                       0
Bank Sta=9734.481,10159.16
Exp/Cntr=0.3,0.1

Type RM Length L Ch R = 1 ,14024.97,240.011000,240.011000,240.011000
XS GIS Cut Line= 6
802534.414823782719864.194127719802501.153007192720015.670475754
802496.642188308720061.209888264802502.479347859720152.685833708
802499.820680331720200.395002353802472.020912502720350.598466853
#Sta/Elev= 30
9738.781106.08769749.891107.98029770.454104.50919780.73598.088119791.016 92.5707
9801.29791.594829832.14192.410949852.61291.906219872.92792.802799883.08591.72213
9913.34790.786529933.44591.457199963.47693.813319973.48888.243469983.543 84.8542
10003.6583.6042110013.69 85.395310023.7287.7684610053.7898.56335 10063.8100.7493
10073.81100.8612   10094102.896710114.24104.140610134.49106.193310154.73 109.186
 10164.9109.725610185.37113.063610205.84115.739910226.31 116.34410232.04117.5602
#Mann= 3 , 0 , 0
9738.781    0.04       09738.781    0.04       010232.04    0.04       0
#XS Ineff= 2 , 0
       09905.794                       0
Bank Sta=9738.781,10232.04
Exp/Cntr=0.3,0.1

Type RM Length L Ch R = 1 ,13784.96,240.010900,240.010900,240.010900
XS GIS Cut Line= 6
802491.225025742719561.684146534802401.093195613719825.921132967
 802361.70851941719926.399251785802327.156265393719992.496550443
802225.010575028720138.689248176802162.217931798720270.923496603
#Sta/Elev= 30
9471.989100.35849486.05898.438249507.18992.007959528.32188.845929560.01888.25654
 9655.1190.625059665.67688.815349697.37388.726099739.63685.850219782.20688.06742
9835.92286.43084  9857.687.499579890.81491.531489925.13892.942119948.84198.93856
9960.916100.44869973.18995.020849985.80183.302699998.41479.5990110022.4883.41922
10035.8994.1141310055.9593.2101910096.2496.9914610119.3798.0655910130.6497.21694
10141.9299.0720310175.2999.7930310197.26 101.02710219.23104.027810258.68105.4256
#Mann= 3 , 0 , 0
9471.989    0.04       09471.989    0.04       010258.68    0.04       0
#XS Ineff= 2 , 0
       09882.569                       0
Bank Sta=9471.989,10258.68
Exp/Cntr=0.3,0.1

Type RM Length L Ch R = 1 ,13544.95,240.011000,240.011000,240.011000
XS GIS Cut Line= 6
802248.270379171719489.747002165802190.207185345 719626.42441165
802147.650470733719733.291619972802109.536193233719834.284765756
802035.226218605720050.324717194 802007.16366915720119.526340923
#Sta/Elev= 30
9487.623 94.93989515.29794.231829547.83687.641919569.52389.30171 9591.2182.93881
9602.05481.161879612.89782.165769634.58481.376839645.35982.742919677.65179.71938
9731.46980.288849774.36178.646469795.73880.073899827.80378.80541 9849.18 80.0301
9880.99877.260289944.41385.027089954.98285.351719965.55284.73121 9986.6976.90508
9997.25976.0397910007.8177.3383310028.9984.6360310039.5889.6209510081.9395.21122
10092.6199.6011110124.99101.970210135.78100.334510146.57102.022410162.24102.6149
#Mann= 3 , 0 , 0
9487.623    0.04       09487.623    0.04       010162.24    0.04       0
#XS Ineff= 2 , 0
       09950.277                       0
Bank Sta=9487.623,10162.24
Exp/Cntr=0.3,0.1

Type RM Length L Ch R = 1 ,13304.94,240.010900,240.010900,240.010900
XS GIS Cut Line= 6
802057.572214477719419.293836062802053.699454691719426.442664401
801986.295557611719563.902754043801826.976041607719909.909387762
801717.382902636720136.060048564801691.654072354720186.376994345
#Sta/Elev= 30
9507.882 85.70739570.09383.729729603.50585.047789669.10984.721879714.36983.12865
9769.43483.943369791.55277.545089824.49973.502899890.57772.963489910.90274.50487
9923.61677.122919956.65588.437069967.66890.634129978.68183.632749989.69472.57758
10000.6972.5086510011.6776.5457910033.6591.76117 10066.891.5463510089.0393.22895
10100.1491.5760110122.3690.2549910133.4891.5552110144.5991.5117810169.2289.68725
10222.38 88.835610266.8386.4603210277.94 87.978310300.1686.9744410357.8588.37658
#Mann= 3 , 0 , 0
9507.882    0.04       09507.882    0.04       010357.85    0.04       0
#XS Ineff= 2 , 0
       09966.987                       0
Bank Sta=9507.882,10357.85
Exp/Cntr=0.3,0.1

Type RM Length L Ch R = 1 ,13064.93,240.011000,240.011000,240.011000
XS GIS Cut Line= 6
802002.205542078719134.723318927801907.556147999719251.108335899
801850.712638018 719335.09902069801807.439206143719406.887204258
801725.982234872 719560.44328543801574.005261662719881.508821168
#Sta/Elev= 30
9264.52279.352739317.42781.011739381.87180.240919419.29678.634099436.99979.68301
 9455.5279.510059491.74578.48843 9503.8277.413939585.95778.079099604.86176.38157
9620.55470.054299625.46269.173249700.08967.732879722.57969.563869834.03270.09139
9900.40573.645529933.59177.789889944.65383.979899955.71586.913089977.83980.40584
9988.901 72.56679999.96369.9041210011.0373.55738 10022.180.8540510033.1682.96634
10077.4384.1528110103.2380.7111710110.6381.56819 10121.785.34224 10128.986.60948
#Mann= 3 , 0 , 0
9264.522  0.0566       09264.522  0.0566       0 10128.9  0.0566       0
#XS Ineff= 2 , 0
       09960.986                       0
Bank Sta=9264.522,10128.9
Exp/Cntr=0.3,0.1

Type RM Length L Ch R = 1 ,12824.92,240.010900,240.010900,240.010900
XS GIS Cut Line= 6
801851.352424524719079.550207458801739.794488164719182.926940936
801673.273397063719259.468837068 801622.95785845719326.504036521
801568.008784025719409.165341757801257.549911286  719913.2327883
#Sta/Elev= 30
9262.41579.534269310.18478.799129350.73780.395259436.67377.512229510.23477.13232
9522.96275.745679547.96965.081529560.47365.119539572.97670.18188 9585.48 71.3229
9650.36671.857959705.91369.895369775.73974.71941 9915.3972.910399939.608 74.4399
9962.38477.984329974.45375.52938   1000166.4104610010.7365.9882410022.8272.09811
10029.58 72.642810047.3869.7818810066.0968.8676410123.9670.5047810143.2567.61586
10162.54 67.240810175.8769.7909210201.1281.9106210210.96 83.107510291.2785.00363
#Mann= 3 , 0 , 0
9262.415  0.0474       09262.415  0.0474       010291.27  0.0474       0
#XS Ineff= 2 , 0
       09952.161        10040.55       0
Bank Sta=9262.415,10291.27
Exp/Cntr=0.3,0.1

Type RM Length L Ch R = 1 ,12584.91,71.646500,71.646500,71.646500
XS GIS Cut Line= 6
801795.539344698719033.889177114801764.861389279719053.724665612
801288.411804825719300.265290633801203.342360407719567.626401767
801116.546217859719844.088189095800754.123610407720134.249665648
#Sta/Elev= 30
9182.82978.440569309.17476.53832 9417.9771.85014 9545.7371.081629590.76865.73928
9602.02765.484549647.06566.731459669.58465.238819700.84366.849669771.28166.86347
9800.05268.136119855.23367.603799876.22168.873879928.69169.483949970.66772.09989
9981.16164.625219997.939 62.995110012.6463.1903910023.1468.7843110033.6371.52487
10131.0173.0935710190.8576.8016810243.2675.7707110264.2278.5311810306.1576.87902
10407.6181.3628210439.6181.14204 10533.1 87.364710725.2592.6462410790.4296.55819
#Mann= 3 , 0 , 0
9182.829  0.0577       09182.829  0.0577       010790.42  0.0577       0
#XS Ineff= 2 , 0
       09944.563                       0
Bank Sta=9182.829,10790.42
Exp/Cntr=0.3,0.1

Type RM Length L Ch R = 2 ,12548.69,,,
Bridge Culvert--1,0,-1,-1, 0
Deck Dist Width WeirC Skew NumUp NumDn MinLoCord MaxHiCord MaxSubmerge Is_Ogee
15.823,40,2.6,0,22,22, , , 0.95, 0, 0,0,,
 9931.38 9933.72 9944.20 9954.34 9954.69 9965.17 9975.65 9986.14 9987.64 9996.62
10007.1110017.5910020.9410028.0710038.5610049.0410054.2410059.5310070.0110080.49
10087.5410088.64
   69.87   70.01   70.63   71.31   71.33   71.77   72.16   72.39   72.40   72.45
   72.49   72.49   72.55   72.71   72.86   72.82   72.84   72.85   72.83   72.86
   72.81   72.82
                                                                                
                                                                                
                
 9931.38 9933.72 9944.20 9954.34 9954.69 9965.17 9975.65 9986.14 9987.64 9996.62
10007.1110017.5910020.9410028.0710038.5610049.0410054.2410059.5310070.0110080.49
10087.5410088.64
   69.87   70.01   70.63   71.31   71.33   71.77   72.16   72.39   72.40   72.45
   72.49   72.49   72.55   72.71   72.86   72.82   72.84   72.85   72.83   72.86
   72.81   72.82
                                                                                
                                                                                
                
BR Coef=-1 , 0 , 0 ,, 0 ,,,0.8,-1,,0,
WSPro=,,,, 1 ,,,, 0 ,,,, 0 ,,,,-1 ,-1 ,-1 , 0 , 0 , 0 , 0 , 0
Multiple Barrel Culv=2,6,11,40,0.013,0.5,1,8,3,64,62,3,Culvert #1, 0, 15.823
 9978.00 9978.0010000.0010000.0010022.0010022.00
Culvert Bottom n=0.013
BC Design=,, 0 ,, 0 ,,,,,,

Type RM Length L Ch R = 1 ,12513.26,224.404300,224.404300,224.404300
XS GIS Cut Line= 6
801643.105566353719005.456520855 801373.04361847719142.652323917
801203.959711552719277.451231733801139.106249273719548.529179528
801053.385763168719802.652443409800638.889235407720081.515290633
#Sta/Elev= 30
9247.03678.202479255.90677.738819266.84975.384329299.67774.978289354.51869.98083
9432.99468.96803 9512.84 69.66299607.86667.078469658.89767.66817 9720.8465.97085
9735.075 62.98489749.31161.929179763.54764.994269785.10963.763169826.30464.50552
9929.29269.573159970.487 69.4532 9980.7462.210969990.97861.6834410021.6962.79615
10031.9371.0395310179.2574.0739910200.3672.2545710284.7971.7404610308.9276.94386
10468.7179.8094610577.1885.3361510661.5587.0749810709.7689.8083710813.5491.56566
#Mann= 3 , 0 , 0
9247.036  0.0714       09247.036  0.0714       010813.54  0.0714       0
#XS Ineff= 2 , 0
       09930.258                       0
Bank Sta=9247.036,10813.54
Exp/Cntr=0.3,0.1

Type RM Length L Ch R = 1 ,12288.86,224.404400,224.404400,224.404400
XS GIS Cut Line= 6
801746.335146762718949.327673307801395.014718706719086.981513555
 801092.40385825719252.169011972801009.188116679719319.552371643
800760.842196807719587.280089264800256.395424405719951.869676281
#Sta/Elev= 30
9090.38776.863859209.07177.706569219.73175.277929251.71175.032959305.13169.43281
9348.16370.253349380.72968.568169478.92269.828779723.71464.727269786.22265.56805
9846.953  62.4539871.82463.03593 9898.7766.028719953.93267.117699966.75366.65581
9978.78462.137819990.81659.4460810014.77  61.63210026.7766.0088910052.4566.52966
10075.2568.9102410134.3971.3212310214.9572.0468710237.9374.7878510307.2577.04343
10345.7277.3719310371.3875.3841510459.6273.7858910669.7775.0213910909.6474.18795
#Mann= 3 , 0 , 0
9090.387  0.0607       09090.387  0.0607       010909.64  0.0607       0
#XS Ineff= 2 , 0
       09867.485                       0
Bank Sta=9090.387,10909.64
Exp/Cntr=0.3,0.1

Type RM Length L Ch R = 1 ,12064.45,224.404300,224.404300,224.404300
XS GIS Cut Line= 6
801744.403529853718940.892339781801099.700374156719167.993379787
800991.803108484719186.745986715800786.118816584719190.181237057
800667.918055058719210.362368017799872.819356948 719464.73288323
#Sta/Elev= 30
9090.05176.731059205.51877.745729216.073 75.0851 9258.2974.389539300.50770.09551
9342.72471.285219527.16468.813389778.54863.29238  9829.860.023929849.94664.20627
9880.16462.705339960.21365.516689970.21565.27866 9990.2258.2906210000.23  57.576
10010.2363.9910310020.2367.2647110100.4468.7227910253.5568.8827910274.2265.73463
10588.5665.8181910641.2863.2253310662.3665.9500510683.45 62.395310715.0861.71074
10746.7163.8704910852.1461.9538110873.2265.2201310936.4864.9810111044.2177.58722
#Mann= 3 , 0 , 0
9090.051  0.0525       09090.051  0.0525       011044.21  0.0525       0
#XS Ineff= 2 , 0
       09816.685        10084.49       0
Bank Sta=9090.051,11044.21
Exp/Cntr=0.3,0.1

Type RM Length L Ch R = 1 ,11840.05,77.111100,77.111100,77.111100
XS GIS Cut Line= 6
801850.911804825718751.654179528800981.120138228718947.834735096
800863.356233507718975.067638054800685.981249273718940.890290633
799911.073794633718943.785800904 798793.91382435718935.528406337
#Sta/Elev= 30
9013.39170.365799101.46169.017769193.72170.653889255.22968.743259306.48569.33548
9326.98767.373669491.00667.444039829.29660.748979911.31461.753549942.10563.85825
9952.36962.038729962.633 57.78719993.42556.7824210003.6957.1012710013.9561.93832
 10044.662.8238310387.5263.4055310627.5360.2472510647.5361.0438110657.5363.99892
10667.5364.3132510897.5364.3759810937.5360.8247911017.5364.0223411107.5359.04463
11297.54 57.703311587.54 59.029811957.5564.6659912047.5663.8622612098.6465.84268
#Mann= 3 , 0 , 0
9013.391  0.0587       09013.391  0.0587       012098.64  0.0587       0
#XS Ineff= 2 , 0
       09684.858        10027.82       0
Bank Sta=9013.391,12098.64
Exp/Cntr=0.3,0.1

Type RM Length L Ch R = 2 ,11800.14,,,
Bridge Culvert--1,0,-1,-1, 0
Deck Dist Width WeirC Skew NumUp NumDn MinLoCord MaxHiCord MaxSubmerge Is_Ogee
16.056,45,2.6,0,55,55, , , 0.95, 0, 0,0,,
 9822.12 9823.88 9828.26 9838.54 9848.82 9859.11 9866.88 9869.39 9873.44 9879.58
 9882.62 9889.72 9899.86 9910.01 9920.15 9930.29 9936.91 9940.48 9950.78 9961.07
 9971.37 9974.81 9981.66 9991.9610002.2510012.5510016.8710022.8410032.7210033.13
10043.2310053.3410059.0510063.4410073.5510083.6510093.7510103.8610113.9610124.07
10128.9410134.1710144.2710154.3810164.4810174.5910184.6910194.7910198.8310204.90
10215.0010225.1110235.2110245.3110254.78
   60.71   60.71   60.69   60.87   60.93   60.80   60.65   60.59   60.64   60.61
   60.53   60.36   60.01   60.30   60.43   60.78   61.20   61.48   62.95   64.13
   64.88   64.95   65.11   65.12   65.04   64.90   64.76   64.53   64.15   64.14
   63.92   63.75   63.64   63.54   63.20   63.11   62.96   62.94   62.84   62.67
   62.62   62.58   62.60   62.60   62.67   62.70   62.69   62.70   62.70   62.68
   62.47   62.01   61.79   61.76   61.73
                                                                                
                                                                                
                                                                                
                                                                                
                                                                                
                                        
 9822.12 9823.88 9828.26 9838.54 9848.82 9859.11 9866.88 9869.39 9873.44 9879.58
 9882.62 9889.72 9899.86 9910.01 9920.15 9930.29 9936.91 9940.48 9950.78 9961.07
 9971.37 9974.81 9981.66 9991.9610002.2510012.5510016.8710022.8410032.7210033.13
10043.2310053.3410059.0510063.4410073.5510083.6510093.7510103.8610113.9610124.07
10128.9410134.1710144.2710154.3810164.4810174.5910184.6910194.7910198.8310204.90
10215.0010225.1110235.2110245.3110254.78
   60.71   60.71   60.69   60.87   60.93   60.80   60.65   60.59   60.64   60.61
   60.53   60.36   60.01   60.30   60.43   60.78   61.20   61.48   62.95   64.13
   64.88   64.95   65.11   65.12   65.04   64.90   64.76   64.53   64.15   64.14
   63.92   63.75   63.64   63.54   63.20   63.11   62.96   62.94   62.84   62.67
   62.62   62.58   62.60   62.60   62.67   62.70   62.69   62.70   62.70   62.68
   62.47   62.01   61.79   61.76   61.73
                                                                                
                                                                                
                                                                                
                                                                                
                                                                                
                                        
BR Coef=-1 , 0 , 0 ,, 0 ,,,0.8,-1,,0,
WSPro=,,,, 1 ,,,, 0 ,,,, 0 ,,,,-1 ,-1 ,-1 , 0 , 0 , 0 , 0 , 0
Culvert=2,4,11,45,0.013,0.5,1,8,3,58,10000,56,10000,Culvert #1, 0, 16.056
Culvert Bottom n=0.013
BC Design=,, 0 ,, 0 ,,,,,,

Type RM Length L Ch R = 1 ,11762.94,328.854200,328.854200,328.854200
XS GIS Cut Line= 6
801809.245138168718689.154179528801159.939582616718824.570846215
800831.758442283718902.741954759800665.147915959718869.709735096
 799872.03882435718854.799239695798845.997157693718849.590906337
#Sta/Elev= 30
9034.83468.038489345.62565.989849366.05561.486619396.701 65.41979519.28366.30098
9703.20760.982679827.037 59.58889921.89759.022489960.69661.822299998.38154.44164
10011.81 54.900410022.0357.5232110032.2662.8695910042.3663.7272310375.91 60.4285
10415.9261.9614210475.9358.3538110585.9557.8709210615.95 60.322510635.9657.71575
10685.97 57.173511026.0257.6500611046.0262.1067411076.02 60.146811236.0259.06973
11296.0256.3849411316.0359.4087911816.0360.8622211956.0365.5394512025.0465.90989
#Mann= 3 , 0 , 0
9034.834  0.0584       09034.834  0.0584       012025.04  0.0584       0
#XS Ineff= 2 , 0
       09611.927        10042.07       0
Bank Sta=9034.834,12025.04
Exp/Cntr=0.3,0.1

Type RM Length L Ch R = 1 ,11434.08,444.106400,444.106400,444.106400
XS GIS Cut Line= 6
802071.397915959718610.595151767801196.397915959718753.824318409
801021.918749303718727.782651767800849.520222038718587.406006813
800786.508662403718571.960746303798877.247157693718815.736739695
#Sta/Elev= 30
 8676.2262.968778692.83662.327828763.76867.262188844.83366.006678905.63168.41098
8976.56367.811819006.962 65.1736 9067.7666.261339341.35461.601129452.81865.00561
 9715.9457.033789901.34859.542419929.05555.943319968.08958.031139998.36753.29564
10028.9360.3928110039.02 60.7215 10069.358.36207 10311.558.2483410372.0555.41927
10543.6155.58441 10553.753.7423410563.7954.2397210573.8958.9661810654.6255.67543
11088.5658.18987 11269.8 56.415111541.6760.0984711722.9259.6061311952.2465.29974
#Mann= 3 , 0 , 0
 8676.22  0.0715       0 8676.22  0.0715       011952.24  0.0715       0
#XS Ineff= 2 , 0
       09481.852        10035.11       0
Bank Sta=8676.22,11952.24
Exp/Cntr=0.3,0.1

Type RM Length L Ch R = 1 ,10989.97,426.633900,426.633900,426.633900
XS GIS Cut Line= 6
802132.777398854718584.739981756801814.348683089718544.894537836
801299.823512018718390.538634315801183.550693721718372.921540633
800748.687412471718388.343994364798890.267991006718742.820073023
#Sta/Elev= 30
8950.43963.99891 9038.36 61.97079118.80266.037839395.06757.280629499.46956.21383
9530.99852.781399730.68552.066049772.65256.784969814.08257.60081 9834.3153.31617
9975.35854.6076210005.3649.2520510035.3657.3551810055.3858.33994 10075.454.11559
10105.4353.4297310205.5254.2102710245.5656.9844410874.8253.33335   1088557.66337
10905.37   54.6511007.1954.2302811322.7957.5761511516.1957.3344711536.5555.77412
11617.9857.8112311689.2455.9419912116.7660.7444312157.4759.54359 12253.964.79985
#Mann= 3 , 0 , 0
8950.439  0.0619       08950.439  0.0619       0 12253.9  0.0619       0
#XS Ineff= 2 , 0
       09796.445        10046.22       0
Bank Sta=8950.439,12253.9
Exp/Cntr=0.3,0.1

Type RM Length L Ch R = 1 ,10563.34,321.162600,321.162600,321.162600
XS GIS Cut Line= 6
802162.607170433718360.855385423801288.820593745718002.473039672
801151.001230717717980.719485715801012.543749273717985.334735081
800363.738851845718112.871877566798911.101324379718677.715906367
#Sta/Elev= 30
8948.63259.708899385.82556.508219396.81356.822319418.78768.031649506.68567.81006
9517.67267.254499528.65958.346229539.64755.26507 9758.8452.199139769.643 48.8284
9780.44650.727079887.39650.45495  9969.353.206749979.34952.923779999.44644.34982
10019.5850.7801510039.6860.8760610109.7253.3708310271.6251.3629710353.1553.49995
 10429.750.3837910750.6152.7118310982.2950.7350410993.0254.6325611014.4752.54723
11143.2351.7578511454.38 55.093611776.2656.3307211840.64  54.77512392.0262.11735
#Mann= 3 , 0 , 0
8948.632  0.0511       08948.632  0.0511       012392.02  0.0511       0
#XS Ineff= 2 , 0
       09682.661        10046.91       0
Bank Sta=8948.632,12392.02
Exp/Cntr=0.3,0.1

Type RM Length L Ch R = 1 ,10242.18,177.555400,177.555400,177.555400
XS GIS Cut Line= 6
802791.222134709717721.677327693 802139.60538125717676.306957304
801462.522047907717751.827790648800516.925399542717876.234928459
800173.582787812718059.858912468798895.476324379718271.465906352
#Sta/Elev= 30
8600.50758.246968616.76957.882688636.81751.459668737.05949.635739308.76347.69475
  9530.6 55.15119741.83556.822719792.04152.663619872.37152.602169922.57746.80816
9952.813 53.09629983.12743.732029993.23243.71748 10134.759.3118110185.2255.62606
10316.4455.11187 10376.950.3444910407.1353.5906810608.6749.03882 11038.553.20166
11208.6152.4950311231.2949.7089311246.7553.7547711554.6253.6123611712.6750.01458
11854.5854.5872711966.0852.0037212229.6258.4130412320.8456.3355412573.7660.76897
#Mann= 3 , 0 , 0
8600.507   0.058       08600.507   0.058       012573.76   0.058       0
#XS Ineff= 2 , 0
       09939.442         10028.4       0
Bank Sta=8600.507,12573.76
Exp/Cntr=0.3,0.1

Type RM Length L Ch R = 3 ,10149.19,,,
BEGIN DESCRIPTION:
END DESCRIPTION:
Bridge Culvert--1,0,-1,-1, 0
Deck Dist Width WeirC Skew NumUp NumDn MinLoCord MaxHiCord MaxSubmerge Is_Ogee
51.777700,74.000000,2.6,0, 60, 60, , , 0.95, 0, 0,0,,
 9716.00 9744.13 9776.40 9804.79 9814.90 9845.22 9915.99 9926.10 9946.32 9961.93
 9961.9310004.9310004.9310048.4510087.8610118.1910148.5210188.9610229.4010252.48
10290.0610320.4910381.0510391.1610431.5510461.8110502.1710537.3810572.7910613.15
10643.4210688.3310724.1310744.3010754.3910764.4810784.6610835.1110855.2810895.64
10905.7310915.8210926.0110936.7310948.1610974.2010990.8811000.2411012.5411034.21
11045.0411066.7011088.3611142.5111182.4811196.6711239.9911250.8211260.5911278.57
   53.84   54.14   54.77   54.71   54.35   54.49   55.25   55.97   55.57   55.55
   55.55   55.65   55.65   55.81   55.53   55.94   55.64   56.10   55.25   55.37
   54.50   54.52   52.90   52.28   51.49   52.23   52.00   52.63   52.31   52.81
   52.48   53.06   52.55   52.96   52.89   53.18   52.74   53.96   53.72   54.36
   54.20   54.29   54.44   54.89   54.59   55.15   54.76   55.14   54.82   54.81
   54.46   54.22   54.20   54.69   54.59   54.91   55.05   55.28   55.17   55.54
 -946.16 -945.86 -945.23 -945.29 -945.65 -945.51 -944.75 -944.03 -944.43 -944.45
   52.55   52.65 -944.35 -944.19 -944.47 -944.06 -944.36 -943.90 -944.75 -944.63
 -945.50 -945.48 -947.10 -947.72 -948.51 -947.77 -948.00 -947.37 -947.69 -947.19
 -947.52 -946.94 -947.45 -947.04 -947.11 -946.82 -947.26 -946.04 -946.28 -945.64
 -945.80 -945.71 -945.56 -945.11 -945.41 -944.85 -945.24 -944.86 -945.18 -945.19
 -945.54 -945.78 -945.80 -945.31 -945.41 -945.09 -944.95 -944.72 -944.83 -944.46
 9716.00 9744.13 9776.40 9804.79 9814.90 9845.22 9915.99 9926.10 9946.32 9969.37
 9969.3710012.3710012.3710048.4510087.8610118.1910148.5210188.9610229.4010252.48
10290.0610320.4910381.0510391.1610431.5510461.8110502.1710537.3810572.7910613.15
10643.4210688.3310724.1310744.3010754.3910764.4810784.6610835.1110855.2810895.64
10905.7310915.8210926.0110936.7310948.1610974.2010990.8811000.2411012.5411034.21
11045.0411066.7011088.3611142.5111182.4811196.6711239.9911250.8211260.5911278.57
   53.84   54.14   54.77   54.71   54.35   54.49   55.25   55.97   55.57   55.57
   55.57   55.66   55.66   55.81   55.53   55.94   55.64   56.10   55.25   55.37
   54.50   54.52   52.90   52.28   51.49   52.23   52.00   52.63   52.31   52.81
   52.48   53.06   52.55   52.96   52.89   53.18   52.74   53.96   53.72   54.36
   54.20   54.29   54.44   54.89   54.59   55.15   54.76   55.14   54.82   54.81
   54.46   54.22   54.20   54.69   54.59   54.91   55.05   55.28   55.17   55.54
 -946.16 -945.86 -945.23 -945.29 -945.65 -945.51 -944.75 -944.03 -944.43 -944.43
   52.57   52.66 -944.34 -944.19 -944.47 -944.06 -944.36 -943.90 -944.75 -944.63
 -945.50 -945.48 -947.10 -947.72 -948.51 -947.77 -948.00 -947.37 -947.69 -947.19
 -947.52 -946.94 -947.45 -947.04 -947.11 -946.82 -947.26 -946.04 -946.28 -945.64
 -945.80 -945.71 -945.56 -945.11 -945.41 -944.85 -945.24 -944.86 -945.18 -945.19
 -945.54 -945.78 -945.80 -945.31 -945.41 -945.09 -944.95 -944.72 -944.83 -944.46
BR Coef=-1 , 0 , 0 ,, 0 ,,,0.8,0,1,0,
WSPro=,,,, 1 ,,,, 0 ,,,, 0 ,,,,-1 ,-1 ,-1 , 0 , 0 , 0 , 0 , 0
BC Design=,, 0 ,, 0 ,,,,,,

Type RM Length L Ch R = 1 ,10064.62,884.885300,884.885300,884.885300
XS GIS Cut Line= 6
802835.492968082717599.281494364802069.177140534717578.911123976
801685.496584982717587.591679558801338.274362683717629.258346215
800485.959547907717757.036123976799285.245040894718064.337092608
#Sta/Elev= 30
8653.95153.142948794.49454.677028944.54746.463139024.57546.521769544.74550.88858
9865.41358.291649875.51258.16025 9895.7148.212869946.20651.749059976.40143.15719
10006.5641.7408510016.6250.3672710026.6752.8277210046.7848.6000210177.5844.89485
10480.3546.7075210530.8150.3250510571.1847.3965810753.0746.5784310956.1350.28651
11048.1947.5169611264.7950.1688411285.4452.5743911306.0847.5532811326.7350.42501
11553.8246.5096211718.9852.3582412173.1654.2340312235.0955.4625412255.4859.36812
#Mann= 3 , 0 , 0
8653.951  0.0448       08653.951  0.0448       012255.48  0.0448       0
#XS Ineff= 2 , 0
       09948.064        10035.22       0
Bank Sta=8653.951,12255.48
Exp/Cntr=0.3,0.1

Type RM Length L Ch R = 1 ,9179.738,595.607100,595.607100,595.607100
XS GIS Cut Line= 6
802876.818470895717550.278617844  802377.5936625717205.357883245
802070.301995844717028.274549916801528.635329127716955.357883245
801059.885329127717059.524549916  800408.8436625717533.482883245
#Sta/Elev= 30
9126.06353.315279208.67855.682369520.41650.027499628.33853.667279679.43852.13694
 9782.3143.550769974.20441.622159990.05939.71112 10001.636.0155610013.1435.70745
10024.6840.5254510034.2942.3342210074.3440.2108910204.1641.0238410426.1438.16027
10771.2639.2226110976.1442.0572111367.9843.6964611405.0942.54133 11442.2 46.1993
11466.9343.1911711514.6445.9654811528.7844.60218   1160345.6762811615.3644.11548
11633.5845.8179411689.5844.6243611887.4948.6270511899.86   50.5811919.8449.19051
#Mann= 3 , 0 , 0
9126.063   0.044       09126.063   0.044       011919.84   0.044       0
#XS Ineff= 2 , 0
       09907.423        10616.33       0
Bank Sta=9126.063,11919.84
Exp/Cntr=0.3,0.1

Type RM Length L Ch R = 1 ,8584.131,493.497400,493.497400,493.497400
XS GIS Cut Line= 6
803539.129657269717111.221897647 802675.53461948716675.668815285
802405.094352663 716565.12624386802244.834711373716484.926441133
  801986.9686625716382.441216573  801096.3436625716377.232883245
#Sta/Elev= 30
 8846.5175.706288950.611 66.5231 8972.7659.337558995.08859.168959006.25255.25981
9084.61756.007529141.00950.817779283.862 51.00169321.46155.512889344.01751.77588
 9389.1351.267819411.68760.699889434.24361.874969468.07849.847769490.63435.77222
9513.19141.486919748.11941.921359791.94136.455479923.51433.309679955.881  33.814
9977.24538.820979987.88337.037759998.522 31.376410019.8338.3966710285.3631.46627
10392.7934.7763910532.6832.8214810894.8136.6839311134.8234.2394811453.4838.68171
#Mann= 3 , 0 , 0
 8846.51   0.041       0 8846.51   0.041       011453.48   0.041       0
#XS Ineff= 2 , 0
       0                10672.47       0
Bank Sta=8846.51,11453.48
Exp/Cntr=0.3,0.1

Type RM Length L Ch R = 1 ,8090.633,493.497500,493.497500,493.497500
XS GIS Cut Line= 6
803672.816396117716672.490277082803106.751961946716373.306386724
802725.325152546716180.641392529802575.663578808716090.362842277
  802236.9686625716002.232883245801309.885329127715944.941216573
#Sta/Elev= 30
8844.52350.607098875.83349.03022  8909.649.347979044.94744.996399067.60542.33422
9101.59342.218179124.25143.972719183.30344.422229247.13741.23994 9310.97 41.1888
9353.52643.225669396.08243.38123 9417.3641.528299430.13732.268789438.63832.00189
9497.99331.71501 9520.4532.893149599.04831.661139889.90630.750689947.55132.42802
9970.90239.418059994.25430.13869   1000129.7310310041.0132.5194910064.3632.58094
10211.6129.6244810335.6129.5511810649.2731.6157511170.2733.0820511365.7536.06454
#Mann= 3 , 0 , 0
8844.523  0.0418       08844.523  0.0418       011365.75  0.0418       0
#XS Ineff= 2 , 0
       0 9717.06        10887.92       0
Bank Sta=8844.523,11365.75
Exp/Cntr=0.3,0.1

Type RM Length L Ch R = 1 ,7597.136,493.497400,493.497400,493.497400
XS GIS Cut Line= 6
803897.089966089716387.932471171803625.568161279716231.159104094
 803398.16255343716083.371455058802875.618802577 715694.11180301
 802533.84366253 715595.98288323  801627.5936625715559.524549901
#Sta/Elev= 30
8829.779 45.22518912.23541.903259050.94741.676569074.21134.188639085.84433.53631
9132.37239.609869192.19237.638039238.74339.939489250.58442.31209 9346.18 40.4649
9370.24635.86863 9446.6134.51497 9467.26 28.24769481.48630.804829516.08731.60165
9584.217 29.22129601.18331.306419615.11728.713099639.93228.459479866.28429.31213
9981.85632.638619991.82232.1462210004.3727.8311910029.4330.6990910171.7330.68867
10316.5827.2047910430.6729.5441211121.2333.8133411191.2931.89988 11328.834.83719
#Mann= 3 , 0 , 0
8829.779  0.0425       08829.779  0.0425       0 11328.8  0.0425       0
#XS Ineff= 2 , 0
       09518.532                       0
Bank Sta=8829.779,11328.8
Exp/Cntr=0.3,0.1

Type RM Length L Ch R = 1 ,7103.638,493.497500,493.497500,493.497500
XS GIS Cut Line= 6
804224.554897815716097.402794555803762.701610684715820.680287361
  803516.0712699715634.588825986803238.377805859 715365.37019138
803065.093662471715273.066216573802122.385329127 715064.73288323
#Sta/Elev= 30
8825.50352.868868996.09949.40587 9030.9352.235579077.37150.139579088.98147.75538
9123.81247.799769191.876 41.07429241.51639.705719320.14443.204739385.99743.22401
9425.34933.188189484.50631.490059509.13434.075729585.25428.841589610.78631.38022
9623.55230.876739636.31826.652369687.97430.873719754.47627.106389767.77628.88077
9895.12926.572499978.64129.06577    999926.29701 10019.829.9156110035.9728.01334
10188.79 26.180910727.8625.9156610840.5128.4403411024.8626.6100111222.1231.00787
#Mann= 3 , 0 , 0
8825.503    0.04       08825.503    0.04       011222.12    0.04       0
#XS Ineff= 2 , 0
       09683.826                       0
Bank Sta=8825.503,11222.12
Exp/Cntr=0.3,0.1

Type RM Length L Ch R = 1 ,6610.141,493.497500,493.497500,493.497500
XS GIS Cut Line= 6
804699.502615392715561.248659909803766.762456387715093.258704782
803231.760329127714882.441216573803070.301995844 714845.98288323
802544.260329127714819.941216573802106.760329127 714877.23288323
#Sta/Elev= 30
8712.56541.952718872.241 40.0433 9095.2345.342669230.42438.436689286.75445.53374
9433.21450.854419550.55470.499359594.72372.773149624.26571.380659680.07358.78131
 9735.88 42.8338 9758.1732.542079769.13930.063649910.31729.674519965.74432.44662
9973.75731.998179994.90321.8880710015.9728.3808410037.03 24.461310058.2228.20231
10087.2325.6816110101.0327.2267510328.7624.3652810421.0926.19083 10843.424.44031
11063.9527.4027611255.5825.2247111366.5230.3287711427.0330.1626411465.59 33.9862
#Mann= 3 , 0 , 0
8712.565  0.0418       08712.565  0.0418       011465.59  0.0418       0
#XS Ineff= 2 , 0
       09838.518                       0
Bank Sta=8712.565,11465.59
Exp/Cntr=0.3,0.1

Type RM Length L Ch R = 1 ,6116.643,493.497400,493.497400,493.497400
XS GIS Cut Line= 6
804919.291698992715137.668306455 804237.66831702714825.056316614
803629.142960548714483.486718908803539.051995844 714455.35788323
803195.301995844 714424.10788323802247.385329127714684.524549901
#Sta/Elev= 30
8692.24529.814218860.63728.93617 8981.1130.597669223.42126.417839635.16326.10953
9736.58424.259689752.08825.558059770.43222.032899815.02321.792359835.60923.28311
9850.419 21.8034  9873.327.014269908.20627.824239979.37327.13241    9999 20.6912
10016.1725.8771210040.4822.6776610072.79 22.004110122.5122.3494810166.1924.94854
10239.3522.7327510279.5123.9663310309.6421.1228610460.2521.0614310550.6323.18669
10798.54 24.468411348.1823.7449711482.99 29.014811524.4829.0624611563.4831.96858
#Mann= 3 , 0 , 0
8692.245  0.0445       08692.245  0.0445       011563.48  0.0445       0
#XS Ineff= 2 , 0
       0 9941.29                       0
Bank Sta=8692.245,11563.48
Exp/Cntr=0.3,0.1

Type RM Length L Ch R = 1 ,5623.146,493.497500,493.497500,493.497500
XS GIS Cut Line= 6
806405.883328375715054.488510869805507.281755463714771.098593134
803895.028086999714088.126949653803674.468662471714038.691216558
803221.343662471714085.566216558802605.477277564  714406.0170185
#Sta/Elev= 30
7419.478 59.6361 7451.4656.694557492.88357.29633 7523.9550.545427679.84337.48683
7794.58133.666288482.10527.023928965.24925.967989321.65521.325569483.90723.10442
9668.09220.407679819.23421.700189841.96829.163269865.44929.901199876.58429.19843
9898.85422.736199943.88622.4627910000.7818.0048710012.1719.0283710023.5624.61813
10046.3521.6660110196.4524.3218510227.1922.0521310268.19      2410309.1821.10538
10410.31 23.819510450.5221.0200910641.5319.8725810701.8521.8983511490.2626.20652
#Mann= 3 , 0 , 0
7419.478  0.0568       07419.478  0.0568       011490.26  0.0568       0
#XS Ineff= 2 , 0
       0 9868.89         10787.5       0
Bank Sta=7419.478,11490.26
Exp/Cntr=0.3,0.1

Type RM Length L Ch R = 1 ,5129.648,493.497400,493.497400,493.497400
XS GIS Cut Line= 6
806549.412700713714497.332256764804569.888594002713798.601662397
803846.343662471713616.816216558803585.926995784 713611.60788323
803247.385329127713715.774549916802669.260329127714054.316216558
#Sta/Elev= 30
7415.687133.61577461.839117.03127482.622112.85967513.79685.962327555.36379.84787
7565.75475.584067774.27761.91483 7858.05 62.22747889.47351.844727910.543 52.0388
7963.21943.368318110.914 30.11648355.27525.53591 8933.8322.160949105.63325.58408
9245.11319.08194 9615.5817.572069698.99218.267599735.38925.482099792.51928.60991
9813.265 18.79769968.85621.017149999.79416.1256410060.8422.0587810091.36 19.3297
10374.3117.5849710434.3221.3056910702.2523.0317311073.9820.1653911547.5724.51211
#Mann= 3 , 0 , 0
7415.687  0.0371       07415.687  0.0371       011547.57  0.0371       0
#XS Ineff= 2 , 0
       09762.211                       0
Bank Sta=7415.687,11547.57
Exp/Cntr=0.3,0.1

Type RM Length L Ch R = 1 ,4636.151,493.497500,493.497500,493.497500
XS GIS Cut Line= 6
806610.915006795714127.928889587805638.471882002713807.793723199
804402.554002622713246.320006121804107.891281209 713158.48288323
803585.926995784 713158.48288323802763.792277298713478.201940419
#Sta/Elev= 30
7411.92793.721347490.77478.832767511.546 63.77967533.81160.369497625.93557.68027
  7678.259.49972 7709.5657.579347730.46648.366497887.79345.933177898.31244.86018
7908.83139.359897940.38736.857527950.90632.021197971.94329.096368035.36426.94489
8157.65329.613898590.84722.254158731.58123.209578927.746 17.22869447.96218.44981
9604.123 15.97819659.89425.083199681.96823.585349692.92118.386079714.82915.78015
9949.97618.3984310001.6915.3904910022.3418.6553810234.8614.7019411506.0524.15315
#Mann= 3 , 0 , 0
7411.927    0.04       07411.927    0.04       011506.05    0.04       0
#XS Ineff= 2 , 0
       09652.175        10542.87       0
Bank Sta=7411.927,11506.05
Exp/Cntr=0.3,0.1

Type RM Length L Ch R = 1 ,4142.654,2588.408700,2588.408700,2588.408700
XS GIS Cut Line= 6
807532.718807131714011.550012887805803.152545393713409.472169191
804757.394026309712992.134324998804025.774362713712613.980568409
803554.676995784712663.691216558802893.218662471 713127.23288323
#Sta/Elev= 30
6730.422138.20146780.946124.68026841.659115.64596902.52784.650777115.56674.87107
7299.75270.85893 7310.3465.636187384.45566.045637419.90756.97103 7458.5754.88692
7857.988 39.07058001.34538.14922 8093.1929.326678238.57430.287648281.15526.29817
8732.47820.363388807.84616.212459721.10916.416659737.78521.839629761.19823.09187
9784.61221.482049796.31915.50855 9831.4413.647459956.169 17.575910012.7414.76369
10053.3518.1605810074.6915.43056 10894.911.97151 11007.617.0854811803.4920.68682
#Mann= 3 , 0 , 0
6730.422  0.0422       06730.422  0.0422       011803.49  0.0422       0
#XS Ineff= 2 , 0
       09760.379        11035.07       0
Bank Sta=6730.422,11803.49
Exp/Cntr=0.3,0.1

Type RM Length L Ch R = 1 ,1554.245,120.227400,120.227400,120.227400
XS GIS Cut Line= 6
805722.213720292 710349.50268133804010.871127695711080.492264688
803211.391961068711304.450598001802578.304754943711414.672522187
800817.835738361711450.332265362800499.576227646711429.761701257
#Sta/Elev= 30
9351.14252.009259359.06344.322039370.04439.724979435.928 31.67619512.79332.01398
9545.73536.993179654.94444.159339754.36829.945879853.1947.3571779897.1179.350868
10006.926.66541910028.8811.0380810066.487.62984610204.586.38933411260.275.015534
11675.67  7.399411785.423.14379912718.919.60237613109.133.86748213319.138.594061
13389.13 8.4265613439.16 -0.559113499.23-0.6561713519.262.38527613669.445.626916
13739.551.65179113759.719.40899313789.9511.0975314090.628.97991714766.7619.61438
#Mann= 3 , 0 , 0
9351.142  0.0426       09351.142  0.0426       014766.76  0.0426       0
#XS Ineff= 2 , 0
       0                12245.52       0
Bank Sta=9351.142,14766.76
Exp/Cntr=0.3,0.1
